--- BLUECR.prj (project) ---

Proj Title=BLUECR
Current Plan=p01
Default Exp/Contr=0,0
English Units
Geom File=g01
Flow File=f01
Plan File=p01
BEGIN DESCRIPTION:
END DESCRIPTION:
DSS Export Rating Curves= 0
DSS Export Rating Curve Sorted= 0
DSS Export Volume Flow Curves= 0
DXF OffsetX= 0
DXF OffsetY= 0
DXF ScaleX= 0
DXF ScaleY= 0

--- BLUECR.p01 (plan) ---

Plan Title=Floodplain
Program Version=4.00
Geom File=g01
Flow File=f01
K Sum by GR=0
Std Step Tol=0.01
Critical Tol=0.01
Num of Std Step Trials=20
Max Error Tol=0.3
Flow Tol Ratio=0.001
Split Flow NTrial=30
Split Flow Tol=0.02
Split Flow Ratio=0.02
Log Output Level=0
Friction Slope Method=1
Unsteady Friction Slope Method=2
Unsteady Bridges Friction Slope Method=1
Global Log Level=0
CheckData=False
Run HTab=0
Run UNet=0
Run PostProcess=0
UNET Theta=0
UNET Theta Warmup=0
UNET ZTol=0
UNET ZSATol=0
UNET MxIter=0
UNET MaxInSteps=0
UNET DtIC=0
UNET DtMin=0
UNET MaxCRTS=0
UNET WFStab=0
UNET SFStab=0
UNET WFX=0
UNET SFX=0
UNET DSS MLevel=0
UNET DZMax Abort=0
UNET Convert EG Bridges=0
UNET Use Existing IB Tables=0
UNET Froude Limit=0
UNET Froude Power=0
Write IC File=0
Echo Input=False
Echo Output=False
Write Detailed=0

--- BLUECR.f01 (steady flow) ---

Flow Title=NFF Regression Equation
Program Version=4.10
Number of Profiles= 1
Profile Names=P100yr
River Rch & RM=BLUECR,Main            ,110648.9
1695.174
River Rch & RM=BLUECR,Main            ,109947
1701.793
River Rch & RM=BLUECR,Main            ,107921.5
1889.406
River Rch & RM=BLUECR,Main            ,105040.2
1955.116
River Rch & RM=BLUECR,Main            ,104621.8
2631.561
River Rch & RM=BLUECR,Main            ,97061.7
2814.906
River Rch & RM=BLUECR,Main            ,96766.4
3197.593
River Rch & RM=BLUECR,Main            ,94126.3
3367.911
River Rch & RM=BLUECR,Main            ,87680.8
3599.784
River Rch & RM=BLUECR,Main            ,85744.5
3840.656
River Rch & RM=BLUECR,Main            ,79154.6
3969.738
River Rch & RM=BLUECR,Main            ,78824.8
5899.687
River Rch & RM=BLUECR,Main            ,67123.3
6295.868
River Rch & RM=BLUECR,Main            ,66856.5
7736.762
River Rch & RM=BLUECR,Main            ,59417.1
8004.664
River Rch & RM=BLUECR,Main            ,46105.7
8368.527
River Rch & RM=BLUECR,Main            ,35603.9
9297.233
River Rch & RM=BLUECR,Main            ,24296.5
9600.324
River Rch & RM=BLUECR,Main            ,10212.3
10016.77
River Rch & RM=BLUECR,Main            ,4820.3
10090.45
River Rch & RM=BLUECR,Main            ,4230.6
10336.28
Boundary for River Rch & Prof#=BLUECR,Main            , 1
Up Type= 0
Dn Type= 1
Dn Known WS=629.1
DSS Import GetInterval= 0
DSS Import GetPeak= 0
DSS Import FillOption= 0

--- BLUECR.g01 (geometry) ---

Geom Title=USGS 10m DEM
Program Version=4.10

River Reach=BLUECR          ,Main
Reach XY= 30
     1896671.507      495150.132     1894848.512      499939.802
     1890079.963      498510.564     1889354.581      496316.247
     1882502.625      496895.942     1877277.226      494614.957
     1870370.611      496587.097     1870477.207      495184.003
     1868439.852      493669.569     1864695.735      494700.904
     1864673.295      496143.535     1861847.157       497406.49
     1862524.095      499397.931     1859381.861      500398.991
     1859850.665      502120.451     1857643.292      500724.443
     1857535.198      503236.078     1854380.907      499618.619
     1852425.999      502589.149      1853592.12      504049.283
     1851624.427      504762.849     1853106.094      506597.849
     1852088.156       508558.08     1849833.992      508920.132
     1849652.808      511052.982     1847310.447      512236.862
     1848597.508      513860.392     1847175.448       514592.27
     1845092.522      521687.356     1841820.127       521648.08

Type RM Length L Ch R = 1 ,110648.9,339.3,335,330.2
XS GIS Cut Line= 2
     1896430.665      495151.717     1896983.087      495171.032
#Sta/Elev= 30
       0 1049.91    48.5 1018.57    58.2    1013    67.9 1010.09    77.6 1008.67
    87.3 1004.76      97  998.58   106.7  992.65   116.4  988.25   126.1  985.84
   135.8  982.14   145.5  975.72   174.6  954.67   184.2  948.08     194  941.97
   213.4  930.39     223  923.21   232.7  916.87   242.4  914.68   252.1   915.9
   261.8   917.6   271.5  918.59     320  920.07   426.7  923.72   436.4  925.04
   446.1  928.13   455.8   932.2   484.9  945.26   523.7  963.12   552.8  976.32
#Mann= 3 , 0 , 0
       0      .1       0   232.7    .045       0   252.1      .1       0
Bank Sta=232.7,252.1
XS Rating Curve= 0 ,0
Exp/Cntr=0.3,0.1

Type RM Length L Ch R = 1 ,110313.9,348.8,366.9,383.9
XS GIS Cut Line= 3
     1896520.391      495500.303     1896676.641      495496.831
     1897065.238      495431.289
#Sta/Elev= 30
       0  978.53     9.8   973.1    19.5  968.39    29.3  965.93    39.1  965.04
    48.8   963.1   107.4  941.25   165.9  920.59   185.1  915.36   198.8  912.42
   204.4  911.54     214  911.36   218.8  911.95   223.6  912.54   233.2   914.9
   242.8   916.3   300.5  917.36   310.1  918.04   319.7  920.37   348.5     932
   358.1  935.39   377.4  941.23     387  943.58   415.8  949.31   454.3   959.5
   463.9  962.41   473.5  966.04   483.1  970.34   492.7  975.21   550.4 1006.76
#Mann= 3 , 0 , 0
       0      .1       0   198.8    .045       0   218.8      .1       0
Bank Sta=198.8,218.8
XS Rating Curve= 0 ,0
Exp/Cntr=0.3,0.1

Type RM Length L Ch R = 1 ,109947  ,392.4,389.7,385.1
XS GIS Cut Line= 3
     1896464.394      495662.339     1896562.822      495704.724
     1897015.244      495998.333
#Sta/Elev= 30
       0  983.04    29.2  971.19      39  966.49    77.9  945.94    87.7  942.36
   107.2  939.71     117   936.8   126.8  933.12   136.6  928.86   156.2  919.16
     166  915.63   175.8  914.53   283.7   911.6   303.3  910.27   313.1  909.71
   322.9  910.66   342.5  916.76   352.3  918.94   381.7  923.94     421  929.78
   430.8  931.79   450.4  937.16     470  943.61   479.8   947.7   489.6  952.53
   509.2  963.25   538.6  977.66   568.1  992.66   636.7 1031.88   646.5 1038.54
#Mann= 3 , 0 , 0
       0      .1       0   303.3    .045       0   322.9      .1       0
Bank Sta=303.3,322.9
XS Rating Curve= 0 ,0
Exp/Cntr=0.3,0.1

Type RM Length L Ch R = 1 ,109557.3,421.3,412.7,402.2
XS GIS Cut Line= 2
     1896303.067      495986.249     1896834.751      496220.624
#Sta/Elev= 30
       0  965.68      29  958.44    87.2  940.58    96.8  938.15   116.2  934.19
   135.6  929.93     155  926.68     213  919.16   242.1  916.28   280.8  913.46
   300.2   911.8   309.9  910.74   313.4  910.13   319.6  909.06   329.3  909.01
   333.4  909.52   348.6  911.14   358.3  911.38   416.4   911.1   435.8   911.2
   445.5  913.19   455.2   918.5   503.6  951.61   513.3  957.43     523  961.75
   532.6  965.72   542.3  969.33   561.7   975.4   571.4  979.04     581   984.3
#Mann= 3 , 0 , 0
       0      .1       0   313.4    .045       0   333.4      .1       0
Bank Sta=313.4,333.4
XS Rating Curve= 0 ,0
Exp/Cntr=0.3,0.1

Type RM Length L Ch R = 1 ,109144.6,344.2,341.8,338.3
XS GIS Cut Line= 2
     1896249.074      496498.879     1896738.657      496498.358
#Sta/Elev= 30
       0  985.11      49  958.78    88.1  937.52    97.9  932.54   117.5   923.6
   137.1  914.85   146.9  911.02   156.7  909.42   166.5  909.62     186  910.44
   215.4  910.98     235  910.79     284   909.8   293.8  909.34   303.5  908.48
   308.6  908.14   313.3  907.82   323.1  907.72   328.6  908.14   332.9  908.46
   342.7  909.81   362.3  912.06   372.1  914.61   381.9  919.05   401.5  928.78
   411.2   933.3   440.6  946.32   450.4  950.45   460.2  954.02   489.6  964.37
#Mann= 3 , 0 , 0
       0      .1       0   308.6    .045       0   328.6      .1       0
Bank Sta=308.6,328.6
XS Rating Curve= 0 ,0
Exp/Cntr=0.3,0.1

Type RM Length L Ch R = 1 ,108802.8,144.5,141.6,139.2
XS GIS Cut Line= 3
     1896405.772      496843.747     1896661.733      496812.313
     1896805.056      496634.979
#Sta/Elev= 30
       0  950.82    19.1  943.44    47.8   931.2    57.3  926.74    66.9  921.94
    76.4  916.71      86  912.04    95.5  909.08   105.1   907.9   114.6  908.22
   116.6  908.47   133.7  910.47   181.5  912.17   238.8  915.56   267.4  916.89
   286.4  917.08   305.4  916.11   314.9  915.96   324.4  916.12   333.9  915.87
   343.4  914.98   352.9  913.73   362.4  913.09   371.9  914.15   381.4   917.6
   390.9   921.7   428.9  939.09   447.9  947.17   466.9  953.75   485.9  959.82
#Mann= 3 , 0 , 0
       0      .1       0    95.5    .045       0   116.6     .06       0
#XS Ineff= 2 , 0
                          284.35           920.4
Permanent Ineff=
       F       F
Bank Sta=95.5,116.6
XS Rating Curve= 0 ,0
Exp/Cntr=0.3,0.1

Type RM Length L Ch R = 1 ,108661.1,42.3,42.3,42
XS GIS Cut Line= 5
     1896423.436      496971.277     1896454.686      496989.507
     1896607.067      496952.314     1896700.052      496832.642
     1896820.137      496685.687
#Sta/Elev= 30
       0  937.72    18.1  932.52    36.2  926.98      46  924.75    65.6  919.27
    75.4  916.96   104.8  911.97   114.6  909.59   118.7  908.91   124.4  907.97
   134.2  907.77   138.7  908.22   153.8  909.96   173.4  910.63   202.5  910.71
   221.4  911.49   259.3  912.62   325.6  916.02   354.1  916.86     373  917.02
     392  916.84   401.5  916.53     411  915.95     430  913.86   439.5  913.31
     449  914.96   458.4  918.34   477.4   925.8   515.4  941.85   534.4  948.65
#Mann= 3 , 0 , 0
       0     .06       0   118.7    .045       0   138.7     .06       0
Bank Sta=118.7,138.7
XS Rating Curve= 0 ,0
Exp/Cntr=0.3,0.1

Type RM Length L Ch R = 1 ,108618.8,110.6,128.4,146.1
XS GIS Cut Line= 5
     1896390.449      497018.152     1896424.554      497039.992
      1896627.59      496989.378     1896749.043      496839.029
     1896877.728      496676.794
#Sta/Elev= 30
       0  935.22    40.5  920.82      69  915.28    88.1  912.42   116.6  909.72
   135.6  908.54   145.1  908.94   155.2  908.37   164.2  907.62   173.7   907.6
   183.2  908.02   202.2  909.46   230.7  915.45   240.2  915.97   249.8   915.5
   269.1  912.17   278.7   911.3   288.4  911.19     385  912.96   452.4  916.18
   508.9  913.37   518.3  913.44   527.7  914.43   537.2   917.8   546.6   922.3
   565.4  932.39   574.8  936.82   584.2   940.5     603  946.64   650.1  959.63
#Mann= 3 , 0 , 0
       0     .06       0   155.2    .045       0   183.2     .06       0
Bank Sta=155.2,183.2
XS Rating Curve= 0 ,0
Exp/Cntr=0.3,0.1

Type RM Length L Ch R = 1 ,108490.4,200.5,213.5,226.3
XS GIS Cut Line= 3
     1896374.824      497039.854     1896695.137      497229.958
     1897011.109      497295.062
#Sta/Elev= 30
       0  931.04    19.6  924.01    39.2  918.03      49  915.38    68.6  911.72
    78.4  909.57    88.2  908.31      98     908   176.4  907.77     196  907.55
   198.9   907.8   215.6  909.43   225.4  909.89   303.9  911.46   323.5  912.22
   343.1  913.39   352.9  914.22   362.7   915.8   372.5  917.94   382.2  919.48
   401.8  921.33   470.2  924.91     480  926.92   548.4  954.24   558.2  958.82
   587.6  976.13   607.1  986.77   626.7  996.79   665.8 1016.03   695.1  1031.4
#Mann= 3 , 0 , 0
       0     .06       0   176.4    .045       0   198.9     .06       0
Bank Sta=176.4,198.9
XS Rating Curve= 0 ,0
Exp/Cntr=0.3,0.1

Type RM Length L Ch R = 1 ,108276.9,343.6,355.4,367
XS GIS Cut Line= 2
     1896281.798      497055.197     1896501.654      497496.715
#Sta/Elev= 30
       0  943.96    19.3  934.99      29  930.58    38.7  926.34    48.4   922.4
      58  919.14    67.7  916.45    77.4  914.93      87   912.4    96.7  908.71
   106.4   907.3   193.4   907.3   203.1  907.54   212.8  907.98   222.4     908
   241.8  907.96     259   907.4   270.8   907.3   280.5  907.34   290.1  907.39
   309.5   907.3   396.5   907.3   406.2     909   415.9  912.48   425.5  916.84
   444.9  925.98   464.2  934.77   473.9  939.39   483.6   944.6   493.2  950.32
#Mann= 3 , 0 , 0
       0     .07       0     259    .045       0   280.5      .1       0
Bank Sta=259,280.5
XS Rating Curve= 0 ,0
Exp/Cntr=0.3,0.1

Type RM Length L Ch R = 1 ,107921.5,275.6,272.5,269.4
XS GIS Cut Line= 2
     1896136.148      497083.105     1896111.158      497550.145
#Sta/Elev= 19
       0  943.79      39  929.08    48.7  925.15    68.2  916.81      78  914.08
    87.7  911.92    97.4  908.93   107.2  907.34   116.9   907.3   282.6   907.3
   302.1   907.3     341  907.33   350.8  908.72   360.5  914.47     380  930.71
   389.8  937.56   399.5  943.02   428.7  958.64   467.7  979.18
#Mann= 3 , 0 , 0
       0    .055       0   282.6    .045       0   302.1      .1       0
Bank Sta=282.6,302.1
XS Rating Curve= 0 ,0
Exp/Cntr=0.3,0.1

Type RM Length L Ch R = 1 ,107649  ,150.2,145.6,141
XS GIS Cut Line= 2
     1895820.702       497057.51     1895862.369      497547.094
#Sta/Elev= 18
       0  952.17    19.6  942.43    39.3  932.52    68.8  918.01    78.6  914.41
    88.4  912.78   108.1   907.3   353.8   907.3   363.6  907.61   373.4  910.89
   383.3   914.7   393.1  918.24   402.9  921.96   412.7  925.96   422.6  930.31
   432.4  934.72   481.5  957.08   491.4  961.48
#Mann= 3 , 0 , 0
       0      .1       0   108.1    .045       0   363.6      .1       0
Bank Sta=108.1,363.6
XS Rating Curve= 0 ,0
Exp/Cntr=0.3,0.1

Type RM Length L Ch R = 1 ,107503.4,133.1,132.2,130.7
XS GIS Cut Line= 3
      1895590.57      497020.556     1895733.972      497498.665
      1895776.53      497597.448
#Sta/Elev= 30
       0  990.71     9.8  985.31    29.4  972.34    39.2  966.22    48.9  961.56
    58.7  957.83    68.5  954.68    78.3  952.43   107.7  947.25   117.4  945.12
   127.2  942.53     137  938.51   146.8  932.07   156.6  924.41   166.4  917.15
   176.2  912.42     186  910.04   195.8  908.12   205.5   907.3   391.5  907.32
   411.1  908.22   420.8  908.12   440.4  907.32   469.8   907.5   479.6  909.01
   489.4  911.98   508.9  919.24   518.7  923.63   557.8  942.14   606.7  962.79
#Mann= 3 , 0 , 0
       0      .1       0   205.5    .045       0   469.8      .1       0
Bank Sta=205.5,469.8
XS Rating Curve= 0 ,0
Exp/Cntr=0.3,0.1

Type RM Length L Ch R = 1 ,107371.2,258.2,237.3,215.9
XS GIS Cut Line= 3
     1895462.109      497091.952     1895625.664      497563.547
     1895672.374      497660.436
#Sta/Elev= 30
       0  981.99    58.7  951.58    88.1  936.75    97.9  932.13     137  915.69
   156.6  906.99   166.4  903.89   176.2  902.06   195.8  900.36   215.3  898.12
   234.9   897.1   264.3  897.46   313.2  900.43   332.8  900.75   342.6  898.04
     350  895.02   352.3  894.08   362.1  893.34   371.9  895.06   401.3  896.52
   440.4  899.06   450.2  900.27     460   902.4   469.8  905.53   479.6  909.81
   499.2   919.9   508.9  924.53   518.7  928.59   557.8  944.17   606.7   962.1
#Mann= 3 , 0 , 0
       0      .1       0     350    .045       0   371.9      .1       0
#XS Ineff= 2 , 0
           326.7   910.8
Permanent Ineff=
       F       F
Bank Sta=350,371.9
XS Rating Curve= 0 ,0
Exp/Cntr=0.3,0.1

Type RM Length L Ch R = 1 ,107133.9,254.9,266.2,276.7
XS GIS Cut Line= 4
     1895037.455      497538.237     1895339.538      497566.883
      1895468.01      497606.813     1895573.913      497702.299
#Sta/Elev= 30
       0  951.32    39.2  938.86    88.1   924.8   107.7  917.57     137  904.41
   146.8  902.27   166.4   901.9   215.3  902.77   225.1  901.85   234.9  899.82
   244.7  898.42   254.5  897.98   303.4  897.96   341.9  897.21   361.1  896.31
   377.7  892.39   380.3  891.68   389.9  891.13   399.5  891.84   409.1  893.88
   418.8  895.26   447.5  896.93   466.5  898.83     476  901.99   485.5  906.59
     514  921.94   523.5  926.62     533  930.56     552  937.11   580.6  945.26
#Mann= 3 , 0 , 0
       0      .1       0   377.7    .045       0   399.5      .1       0
#XS Ineff= 2 , 0
          300.85  902.13
Permanent Ineff=
       F       F
Bank Sta=377.7,399.5
XS Rating Curve= 0 ,0
Exp/Cntr=0.3,0.1

Type RM Length L Ch R = 1 ,106867.7,186,169.6,152.6
XS GIS Cut Line= 3
     1895101.995      497673.435     1895279.078      497792.358
      1895423.61       497936.89
#Sta/Elev= 30
       0  923.01    38.8  910.86    67.9  901.46    77.6  899.04    87.3  898.31
   155.1  895.17   164.8  894.54   174.5  893.43   184.2  891.71   203.6  892.45
   213.3  892.41     223  891.71   237.1  889.71   242.5  888.98   252.2  889.01
   257.1  889.75     262  890.49   271.7  892.42   281.4  893.19   291.2  893.68
   300.9  894.68   310.6  897.16   320.4  901.02   330.1  905.84   349.6  915.87
   359.3  920.42     369  924.11   378.8  927.09   398.2  932.59   417.7  938.48
#Mann= 3 , 0 , 0
       0      .1       0   237.1    .045       0   257.1      .1       0
Bank Sta=237.1,257.1
XS Rating Curve= 0 ,0
Exp/Cntr=0.3,0.1

Type RM Length L Ch R = 1 ,106698.2,331.6,330.8,329.5
XS GIS Cut Line= 3
     1894979.462      497939.082     1895314.144      497955.623
     1895414.415       497977.97
#Sta/Elev= 30
       0  935.81     9.6  930.38    19.2   925.4    28.7  921.23    38.3  917.88
    47.9  915.16    57.4  913.15    76.6   911.6    86.2  909.88    95.7   906.6
   105.3  901.75   114.9  895.87   124.5  891.95     134  891.42   143.6  892.14
   153.2  892.34   172.3  891.66   191.5  890.37   210.6   888.2   220.2  887.22
   229.8  886.83   248.9  887.53   315.9  892.63   335.1  894.44   344.4  897.22
   353.8  901.89   372.4  912.69   391.1  921.12   409.8  928.61   437.8  938.36
#Mann= 3 , 0 , 0
       0      .1       0   210.6    .045       0   248.9      .1       0
Bank Sta=210.6,248.9
XS Rating Curve= 0 ,0
Exp/Cntr=0.3,0.1

Type RM Length L Ch R = 1 ,106367.4,248.6,252.3,254.7
XS GIS Cut Line= 5
     1894963.348       498284.32     1895145.192      498272.419
     1895145.717      498272.393     1895337.208      498273.768
     1895492.862      498287.793
#Sta/Elev= 30
       0  937.57    38.4  925.51      48  923.63    86.3  920.52   115.1   917.8
   143.9  913.83     163  910.65   172.6  908.67   182.8  906.06   192.3  902.34
   211.5  892.12   221.1  890.64   240.2  890.52   249.8  889.72   288.1  885.14
   297.7  884.49   307.2  884.83   308.9  885.14   316.8  886.58   345.5  894.84
   364.7  899.69   374.2  902.46     384  906.85   393.8  912.91   403.6  920.75
   423.1   941.2   432.9   949.1   442.6     955   471.9  971.96   530.5 1007.76
#Mann= 3 , 0 , 0
       0      .1       0   288.1    .045       0   308.9      .1       0
Bank Sta=288.1,308.9
XS Rating Curve= 0 ,0
Exp/Cntr=0.3,0.1

Type RM Length L Ch R = 1 ,106115.1,244.3,250.2,255.8
XS GIS Cut Line= 2
      1895041.69      498490.701     1895409.529      498541.699
#Sta/Elev= 28
       0  901.27     9.8  898.23    19.6  895.36    29.3  893.45    39.1  892.81
    78.2  891.69    97.7  891.24   107.5  890.67   117.3  889.02     127   886.7
   136.8  883.96   146.6  881.52   156.4  880.82   166.1  881.12   175.9  882.08
     215  885.96   234.5  888.28   244.3  891.51   254.1  897.89   263.9  905.43
   283.4  921.62   312.7   946.6   322.5   954.6   332.3  962.39     342  969.74
   351.8  976.27   361.6  982.05   371.4  987.57
#Mann= 3 , 0 , 0
       0      .1       0   146.6    .045       0   175.9      .1       0
Bank Sta=146.6,175.9
XS Rating Curve= 0 ,0
Exp/Cntr=0.3,0.1

Type RM Length L Ch R = 1 ,105864.9,274.6,272.5,270.4
XS GIS Cut Line= 2
     1895006.214      498670.936     1895310.752      498799.201
#Sta/Elev= 27
       0  901.04    19.4  893.67    29.2  890.64    38.9  889.11    48.6  888.91
    87.5   888.9    97.2  888.69   106.9  887.96   116.6  886.89   155.5  882.06
   165.2  880.81   174.9  879.38   177.1  879.16   184.7  878.39   194.4   878.3
   197.1  878.88   204.1  880.37   213.8  884.03   233.3   891.1     243  895.52
   252.7   900.7   262.4  905.76   291.6  920.76   301.3  925.97     311  931.48
   320.7  937.27   330.4  943.39
#Mann= 3 , 0 , 0
       0      .1       0   177.1    .045       0   197.1      .1       0
Bank Sta=177.1,197.1
XS Rating Curve= 0 ,0
Exp/Cntr=0.3,0.1

Type RM Length L Ch R = 1 ,105592.3,238.4,232,224.4
XS GIS Cut Line= 3
     1894938.913      498951.855     1895191.423      499031.699
     1895315.302      499048.383
#Sta/Elev= 30
       0  911.67    19.6  904.06      49  892.41    58.8  888.77    68.7   886.7
    78.5  886.34    88.3  886.53    98.1  885.96   107.9  884.06   117.7  881.23
   127.9  878.85   137.3  878.03   147.9  878.34   176.6  880.56   196.2  881.82
   235.4  884.07   245.2  885.77     255   889.5   264.8  894.44   274.4  899.46
   303.3  913.98   312.9  918.89   322.5  923.93   332.1  929.17   341.8  934.66
   351.4   940.4     361  946.33   370.6   952.4   380.2  958.77   389.8  965.43
#Mann= 3 , 0 , 0
       0      .1       0   127.9    .045       0   147.9      .1       0
Bank Sta=127.9,147.9
XS Rating Curve= 0 ,0
Exp/Cntr=0.3,0.1

Type RM Length L Ch R = 1 ,105360.4,317.1,320.2,322.3
XS GIS Cut Line= 3
     1894812.611      499175.727     1894921.552       499208.32
     1895278.775      499208.496
#Sta/Elev= 30
       0  936.95    28.4  923.16    37.9   919.3    47.4  915.79    56.9   912.6
    66.3   909.7     133  889.93   152.3  884.46     162  882.89   171.6  882.45
   181.3  881.77   200.6  878.06   210.3  877.22   219.9  877.23   229.6  878.14
   248.9  881.09   258.5   882.3   268.2  883.14   277.8  883.53   287.5  883.64
   297.2  883.49   316.5   882.8   326.1  882.71   335.8  883.11   345.4  885.44
   355.1  890.13   393.7  912.72   422.7  930.22     442   942.1   470.9  960.18
#Mann= 3 , 0 , 0
       0      .1       0   200.6    .045       0   229.6      .1       0
Bank Sta=200.6,229.6
XS Rating Curve= 0 ,0
Exp/Cntr=0.3,0.1

Type RM Length L Ch R = 1 ,105040.2,165.8,166.8,167.9
XS GIS Cut Line= 4
     1894828.872      499493.414     1894945.192      499509.039
     1895158.733      499535.514     1895279.827      499487.337
#Sta/Elev= 30
       0  922.85     9.8  919.33    19.6   915.2    29.3  910.91    39.1  906.73
    58.7  898.59    68.5  894.42      88  885.67    97.8  882.44   107.6  881.55
   117.4  881.73   127.1  881.04   136.9  879.28   146.7  877.17   156.5  875.67
   166.3  875.35     176  875.83   185.8  876.58   195.6  877.16   205.4  877.61
   234.7  878.65   254.3  879.17   283.6  880.12     313  881.29   322.8  882.02
   332.5   884.4   379.1  902.92   388.4  906.99   397.7  911.75   462.9  949.72
#Mann= 3 , 0 , 0
       0      .1       0   156.5    .045       0     176      .1       0
Bank Sta=156.5,176
XS Rating Curve= 0 ,0
Exp/Cntr=0.3,0.1

Type RM Length L Ch R = 1 ,104873.3,235.7,251.5,265.8
XS GIS Cut Line= 4
     1894791.192       499555.77     1894880.602      499663.409
     1895120.185      499704.207     1895315.498       499560.11
#Sta/Elev= 30
       0   928.3     9.3  926.19    18.7  923.47      28  919.28    37.3  913.98
    46.6  908.18    74.6  889.25      84  884.06    93.3  881.56   111.9  881.98
   121.3  881.67   188.5  877.79   236.6  874.26   246.9  873.96   256.6  874.21
   305.2  878.05   324.6  879.32   344.1  880.16   363.5  880.68   402.4  881.37
   460.6  881.93   470.3  882.52     480   884.6   489.8  888.59   538.3   910.6
   557.7   918.8   567.4  923.32   577.1  928.39   596.6  939.57   625.7  954.85
#Mann= 3 , 0 , 0
       0      .1       0   236.6    .045       0   256.6      .1       0
Bank Sta=236.6,256.6
XS Rating Curve= 0 ,0
Exp/Cntr=0.3,0.1

Type RM Length L Ch R = 1 ,104621.8,418,439.9,460.7
XS GIS Cut Line= 5
     1894753.267      499563.785     1894854.378      499860.451
     1894944.934       499954.34     1894981.375      500051.774
     1895131.253      500196.178
#Sta/Elev= 30
       0  934.49    29.4  927.42    39.2   924.5      49  920.35    58.8  914.62
    97.9  885.46   107.7  881.51   137.1  881.24   264.4  874.71   322.7  872.69
   372.7  873.15   392.7  872.89   415.9  873.57   453.3  873.33   462.8  873.82
   472.2  878.32   481.7  887.23   491.2  895.38   500.6  901.32   547.9  929.43
   576.3  944.42   595.2  954.93   623.6  972.16   642.5  984.82     652  991.62
   708.7 1033.68   727.6 1046.77   737.1 1052.81   746.6 1057.05     756 1057.83
#Mann= 3 , 0 , 0
       0      .1       0   372.7    .045       0   392.7      .1       0
Bank Sta=372.7,392.7
XS Rating Curve= 0 ,0
Exp/Cntr=0.3,0.1

Type RM Length L Ch R = 1 ,104181.9,433.8,462.4,491.4
XS GIS Cut Line= 3
     1894543.395      499633.096     1894470.478      500021.985
     1894559.888      500263.304
#Sta/Elev= 30
       0  928.87      29  919.48    38.6  915.96    48.2  911.14    57.9  903.09
    67.6   892.6    77.2  884.15    86.8  880.54    96.5  879.78   164.1  876.48
   289.5  871.31   308.8  871.16   318.5  871.63   328.1  875.32   337.8  881.59
   347.4  886.32     386  895.19   395.7  897.07   405.2  899.26   424.3  902.82
   443.3  905.56   452.8  907.94   462.4  911.28   471.9   915.5     510  933.28
   538.6  948.32   548.2  952.17   557.7  955.35     634  978.88     653  985.01
#Mann= 3 , 0 , 0
       0      .1       0   289.5    .045       0   318.5      .1       0
Bank Sta=289.5,318.5
XS Rating Curve= 0 ,0
Exp/Cntr=0.3,0.1

Type RM Length L Ch R = 1 ,103719.4,346.3,336.7,326.2
XS GIS Cut Line= 4
     1894445.575       499519.11     1894298.353      499646.332
     1894076.686      499670.776     1893861.409      499809.145
#Sta/Elev= 30
       0  952.84     9.7  945.69    19.5  939.19    29.2  933.94    38.9  930.46
    48.6  927.94     107  915.01   116.8  912.39   126.5  903.61   136.2  890.69
   145.9  880.11   155.7  876.55   184.8  874.78   268.8870.9803   281.8  870.49
   291.3  870.53   301.2  871.33   320.6   873.8   417.6  879.23   455.5  880.76
     465  881.67   474.5   883.9   483.9  887.53   540.8   911.8   559.8  920.71
   578.7  930.27   607.2  945.48   626.1  956.27   645.1  967.69   673.5  985.66
#Mann= 3 , 0 , 0
       0      .1       0   268.8    .045       0   301.2      .1       0
Bank Sta=268.8,301.2
XS Rating Curve= 0 ,0
Exp/Cntr=0.3,0.1

Type RM Length L Ch R = 1 ,103382.7,495.7,493.3,490.1
XS GIS Cut Line= 2
     1894271.344      499250.631     1893814.023      499536.076
#Sta/Elev= 30
       0  948.57    39.2  924.44      49  919.61    58.8  916.36    88.2  908.33
      98  904.54   107.8  896.63   117.6  885.79   127.4  877.95   137.2  875.14
     147  873.77   156.8  871.14   166.6  869.11   176.4  869.04   186.2  870.13
     196  871.34   205.8  872.03   254.8  873.89   303.8  876.68   382.3  882.52
   421.5  885.64   431.3  886.59   441.1  888.73   450.9  892.04   470.5  899.32
   499.9  909.96   509.7  913.89   519.5  918.13   529.3  922.68   539.1  927.48
#Mann= 3 , 0 , 0
       0      .1       0   156.8    .045       0   186.2      .1       0
Bank Sta=156.8,186.2
XS Rating Curve= 0 ,0
Exp/Cntr=0.3,0.1

Type RM Length L Ch R = 1 ,102889.5,484.7,472.9,460.8
XS GIS Cut Line= 2
     1893921.532      498915.576     1893555.559      499241.964
#Sta/Elev= 30
       0  914.59    19.6   907.7    29.4  905.16    39.2  903.88    88.3   898.7
   117.7  895.77   147.1  893.27   156.9  891.24   166.7  886.24   176.5  877.95
   186.3  872.36   196.2  869.86   215.8  865.99   225.6  864.55   235.4  864.43
   245.2  866.02     255  868.35   264.8  869.99   274.6  870.58   353.1  871.57
   362.9  871.82   372.7  873.01   382.5   876.2   402.1  884.59   441.3   900.4
   451.1  904.62     461  909.12   470.8     914   480.6  919.14   490.4   924.5
#Mann= 3 , 0 , 0
       0      .1       0   215.8    .045       0   245.2      .1       0
Bank Sta=215.8,245.2
XS Rating Curve= 0 ,0
Exp/Cntr=0.3,0.1

Type RM Length L Ch R = 1 ,102416.6,505.1,488.3,470.7
XS GIS Cut Line= 3
     1893497.052      498565.749     1893352.788      498803.854
     1893267.886      499030.333
#Sta/Elev= 30
       0  917.15     9.6   913.1    19.2  909.34    28.8  906.11    38.4  903.36
      48  900.89    57.6  898.69      96  891.13   105.6  889.12   115.2   886.1
   124.8  881.15   134.4  875.13     144  871.55   153.6  870.54   163.2  870.21
   182.4  869.94   201.6  869.34   220.8  868.49   259.2  867.29   307.4  865.54
   336.4  864.04   346.1  863.54   355.8  863.41   365.5  863.99   384.8   866.8
   404.2   869.2   413.8  870.87   423.5  873.36   462.2  886.11   520.3  904.86
#Mann= 3 , 0 , 0
       0      .1       0   336.4    .045       0   365.5      .1       0
Bank Sta=336.4,365.5
XS Rating Curve= 0 ,0
Exp/Cntr=0.3,0.1

Type RM Length L Ch R = 1 ,101928.3,317.8,318.6,319.3
XS GIS Cut Line= 2
     1892858.382      498635.173     1893055.489       499102.32
#Sta/Elev= 30
       0  898.94     9.8  897.35    19.5  896.21    29.2  895.29      39  894.09
    48.8  892.17    58.5  888.28    68.2  882.52      78  876.38    87.8  871.19
    97.5  868.08   107.3  865.33   113.2 863.335     117  862.05   126.8  860.04
   136.5  860.18   146.3  862.35     156  865.79   165.8  867.91   175.5  868.69
   224.3  870.41   253.5  871.66   341.3  876.22     351  877.02   360.8  878.71
     390  886.37   458.3  903.36     468  905.85   487.5  911.15     507  916.84
#Mann= 3 , 0 , 0
       0      .1       0   113.2    .045       0   146.3      .1       0
Bank Sta=113.2,146.3
XS Rating Curve= 0 ,0
Exp/Cntr=0.3,0.1

Type RM Length L Ch R = 1 ,101609.7,207.7,205.1,201.8
XS GIS Cut Line= 4
     1892577.132      498675.798     1892578.834      498783.136
     1892638.382      498938.923     1892750.049      499200.798
#Sta/Elev= 30
       0  910.89     9.8  905.88    19.5  901.34    29.3  897.55      39  894.53
    48.8  891.95    58.6  889.69    68.3  887.88    78.1  886.64   107.4  884.31
   117.2  883.04     127  881.08   136.8   877.6   156.4  866.85   166.2  864.53
     176  863.12   185.8  861.18   195.6  859.08   205.5  857.93   215.3  858.39
   225.1  861.23   234.9  864.97   244.7  867.08   254.5  867.77   303.6   870.2
   372.3  872.95   411.6  874.85   431.2  876.37   490.1  882.21   558.8  888.44
#Mann= 3 , 0 , 0
       0      .1       0   185.8    .045       0   225.1      .1       0
Bank Sta=185.8,225.1
XS Rating Curve= 0 ,0
Exp/Cntr=0.3,0.1

Type RM Length L Ch R = 1 ,101404.6,477.5,510.8,543.3
XS GIS Cut Line= 4
     1892392.757      498691.076     1892386.681      498831.701
     1892494.858      499029.742     1892572.445      499283.089
#Sta/Elev= 30
       0  902.75    37.5  887.17    56.3   879.8    65.7  876.36    75.1  873.15
    84.4  870.27    93.8  868.37   103.2  867.56   150.6  866.34   170.2  865.37
     180  864.38   189.8  862.71   202.8859.5515   209.4  858.09   219.2  857.22
   229.1  857.39   238.9  858.27   268.3  861.05   297.7  863.43   405.7  869.88
   474.4  874.24   484.2  875.02   503.8  876.93   533.2  880.13   552.9  882.59
   582.3  887.12   592.1  888.77   601.9  891.09   611.8  894.52   631.4  902.92
#Mann= 3 , 0 , 0
       0      .1       0   202.8    .045       0   238.9      .1       0
Bank Sta=202.8,238.9
XS Rating Curve= 0 ,0
Exp/Cntr=0.3,0.1

Type RM Length L Ch R = 1 ,100893.8,504.7,473.1,439.8
XS GIS Cut Line= 4
     1892112.337      498641.349       1892088.9      498891.349
     1891942.198      499000.724     1891977.789      499220.342
#Sta/Elev= 30
       0  904.82    77.3  875.83    86.9  873.65   106.2  873.25   115.9  869.89
   125.6  865.62   135.2  862.56   144.9  861.41   173.8  860.15   299.2  857.12
   318.5   856.9   328.1   857.4   337.8  859.38     357   864.7   366.7  866.25
   385.9  867.65   424.4  868.96   434.1  869.76   443.8  871.86   453.4  875.67
   482.4  891.46   492.1   895.9   511.5  903.11   550.2  914.76   569.5  921.41
   579.2  925.97   608.2  942.32   627.6  951.71   646.9   958.6   656.6   960.6
#Mann= 3 , 0 , 0
       0      .1       0   299.2    .045       0   337.8      .1       0
Bank Sta=299.2,337.8
XS Rating Curve= 0 ,0
Exp/Cntr=0.3,0.1

Type RM Length L Ch R = 1 ,100420.7,432.7,462.1,490.6
XS GIS Cut Line= 3
     1891621.765      498743.182     1891657.911      498883.356
     1891790.133      499135.022
#Sta/Elev= 30
       0  892.96     9.6  889.65    19.3  886.78      29  884.66    38.6   883.2
    67.6  879.59   115.8  874.65   125.5  874.14   135.1  873.22   144.8  870.65
   154.6  867.02   164.4  863.88   174.2  862.22   223.2  859.68   237.2857.7971
   242.8  856.86   252.6  855.92   262.4  856.53   267.2857.5831   272.2  858.68
   291.8  863.71   311.4   867.9   321.2  869.64   340.8  872.48   350.6   874.2
   360.4  876.46     380  881.69   399.6  887.38   409.4  890.34     429  896.72
#Mann= 3 , 0 , 0
       0      .1       0   237.2    .045       0   267.2      .1       0
Bank Sta=237.2,267.2
XS Rating Curve= 0 ,0
Exp/Cntr=0.3,0.1

Type RM Length L Ch R = 1 ,99958.7 ,411.7,396.7,382
XS GIS Cut Line= 4
     1891505.793       498708.46     1891499.179      498792.099
     1891280.119      499006.029     1891220.675      499167.279
#Sta/Elev= 30
       0  910.36     9.3  906.35      28  898.84    55.9  888.48    74.6   882.1
     103  872.73   122.2  866.74   131.7  864.14   141.3  862.56   150.9  862.04
   179.6  861.79   265.7  860.05   275.3  859.55   288.7857.3478   294.4  856.38
     304  855.87   313.5  856.62   318.7857.8279   323.1  858.85   332.7  861.79
   351.8  868.62   361.4  871.82     371  874.34   380.5   876.3   409.2  881.56
     476  893.45   485.6  895.34   514.2  902.82   552.4  911.99     562  914.66
#Mann= 3 , 0 , 0
       0      .1       0   288.7    .045       0   318.7      .1       0
Bank Sta=288.7,318.7
XS Rating Curve= 0 ,0
Exp/Cntr=0.3,0.1

Type RM Length L Ch R = 1 ,99562   ,408.8,413.5,417.6
XS GIS Cut Line= 2
     1891059.968      498567.684     1890990.981      499080.251
#Sta/Elev= 30
       0  928.02    29.3  908.59    68.3   881.9    87.8  868.89    97.6  863.37
   117.1  855.88     119855.3484   126.9  853.14   136.6  852.87   146.4  854.17
     149854.7088   156.1  856.18   165.9  857.97   175.6  859.06   185.4  859.35
   224.4  859.18   253.7  858.82   273.2  858.82   292.8  859.19   302.5   859.2
   312.3  859.48   331.8  860.27   341.5   861.2   351.3  863.23   390.3  873.39
   419.6  881.63   458.6  892.87   478.2  898.25   497.7  903.78   517.2   909.6
#Mann= 3 , 0 , 0
       0      .1       0     119    .045       0     149      .1       0
Bank Sta=119,149
XS Rating Curve= 0 ,0
Exp/Cntr=0.3,0.1

Type RM Length L Ch R = 1 ,99148.5 ,322.8,327.4,331.5
XS GIS Cut Line= 3
     1890682.371      498544.344     1890612.859      498748.535
     1890491.031        498940.4
#Sta/Elev= 30
       0  896.24    19.6  887.74    39.2   879.6    58.8  871.79    78.4  864.67
    88.2  861.91      98  859.86   107.8  858.79   117.6  858.43   127.5  857.67
   137.3  855.58   143.6853.8893   147.1  852.95   156.9  851.74   166.7  852.52
   173.6854.6463   186.3  858.66   196.1  860.36   205.9  861.48   215.7  862.09
   234.6  862.45     263  862.05     282  862.15   310.4  862.71   319.9  863.39
   329.3   865.9   348.3  873.86   357.8  877.58   367.2  880.87     443  906.38
#Mann= 3 , 0 , 0
       0      .1       0   143.6    .045       0   173.6      .1       0
Bank Sta=143.6,173.6
XS Rating Curve= 0 ,0
Exp/Cntr=0.3,0.1

Type RM Length L Ch R = 1 ,98821.1 ,351,376.2,400.3
XS GIS Cut Line= 2
     1890413.266      498441.264     1890231.365      498759.285
#Sta/Elev= 23
       0  887.98    28.9  875.29    57.8  862.82    67.5  859.44    77.1  857.61
    86.8  856.02    96.4  853.43     106   851.6   115.7  852.15   124.2853.6282
   125.3  853.82     135  854.88   144.6  855.26   173.5  855.69     241  856.88
   250.7  857.34   260.3  860.12     270  865.84   279.6  872.38   289.2  877.67
   298.9  881.59   327.8  892.13   366.4  905.34
#Mann= 3 , 0 , 0
       0      .1       0    96.4    .045       0   124.2      .1       0
Bank Sta=96.4,124.2
XS Rating Curve= 0 ,0
Exp/Cntr=0.3,0.1

Type RM Length L Ch R = 1 ,98444.9 ,350.6,338.9,326.5
XS GIS Cut Line= 4
      1890285.09      498315.747     1890111.046      498432.425
     1889932.627      498427.077     1889745.385      498493.689
#Sta/Elev= 30
       0  909.56    38.1  893.53    57.2  882.43    66.7  878.24    85.7  873.74
    95.2  870.43   114.3  862.12   123.8  858.46   133.3  856.86   142.9  856.53
   209.5  855.92   237.7   855.1   247.1     854   255.3852.4036   265.9     851
   275.3  851.64   284.7  854.37   294.1  857.79   303.5  860.01   341.1  863.19
   350.5  865.26     388  878.94     407   884.8   444.8  894.18   511.1  909.09
   520.5  911.96   539.4  919.53   558.4     928   577.3  935.78   586.8  940.27
#Mann= 3 , 0 , 0
       0      .1       0   255.3    .045       0   284.7      .1       0
Bank Sta=255.3,284.7
XS Rating Curve= 0 ,0
Exp/Cntr=0.3,0.1

Type RM Length L Ch R = 1 ,98106   ,521.3,524,524.8
XS GIS Cut Line= 2
     1890108.936      498043.209     1889705.455      498264.464
#Sta/Elev= 30
       0  913.07    29.4  899.67      49  891.03    58.7  886.31    78.3  876.34
    88.1  870.02   107.7  858.17   117.5  854.23     135850.5914   137.1  850.15
   146.9  849.38   156.6  850.19     165851.6899   176.2   853.1     186  853.29
   244.8  853.52   274.1  854.16   283.9  854.78   293.7  857.82   303.5  863.24
   313.3   869.5   323.1  875.08   332.9  878.95   342.7  882.02   352.5  884.42
     372  889.71   381.8  893.11   391.6  897.36   411.2   906.4   460.2  927.02
#Mann= 3 , 0 , 0
       0      .1       0     135    .045       0     165      .1       0
Bank Sta=135,165
XS Rating Curve= 0 ,0
Exp/Cntr=0.3,0.1

Type RM Length L Ch R = 1 ,97582   ,509.6,520.3,530.6
XS GIS Cut Line= 3
     1889897.434       497655.08     1889604.251      497781.347
     1889420.499      497832.897
#Sta/Elev= 30
       0  923.41    19.4  916.61      29  912.97    38.7  908.84    48.4  904.33
      58  899.51    77.4  889.04   116.1  866.05   125.8  860.54   135.4  856.26
   155.4849.4052   164.4  847.38   174.1  847.57   185.4849.5489   193.5  850.91
   203.1  851.96   212.8   852.6   251.5  854.36   270.8  856.16   299.9  860.32
   309.5  862.04   328.8  866.78   338.3  869.51   347.8  872.62   376.5  883.27
   395.6  890.62   443.3  910.79   452.8  914.56     491  928.31   510.1  935.41
#Mann= 3 , 0 , 0
       0      .1       0   155.4    .045       0   185.4      .1       0
Bank Sta=155.4,185.4
XS Rating Curve= 0 ,0
Exp/Cntr=0.3,0.1

Type RM Length L Ch R = 1 ,97061.7 ,291.9,295.3,298.6
XS GIS Cut Line= 3
     1889919.862      497349.483     1889703.735       497312.57
     1889377.382      497297.683
#Sta/Elev= 30
       0  952.61     9.5  949.44    28.6  943.65    47.7  937.63    66.7  931.92
    76.3  928.85    85.8  925.44   123.9  911.15   162.1  897.16   171.6  893.51
   181.1  889.69   190.7  885.69   219.3   873.2   248.1  860.34   257.7  856.59
   267.3  854.35   276.9  853.54   344.2  852.28   411.4  850.09     421  849.51
   431.7848.1844   440.2  847.14   449.9  847.31   459.5  851.47   478.7   865.7
   488.3  872.08   497.9  878.02   507.5  883.41   517.1  888.39     546  902.95
#Mann= 3 , 0 , 0
       0      .1       0   431.7    .045       0   459.5      .1       0
Bank Sta=431.7,459.5
XS Rating Curve= 0 ,0
Exp/Cntr=0.3,0.1

Type RM Length L Ch R = 1 ,96766.4 ,135.3,130.6,125.8
XS GIS Cut Line= 5
     1890031.124      497039.899     1889790.847      497028.787
     1889632.513      497032.954      1889455.43      496998.232
     1889396.402      496998.926
#Sta/Elev= 30
       0  859.63    67.4     858   125.1   856.9   163.6  855.85   240.5  855.64
   268.5  855.27   305.8  854.44   333.7  854.12   352.3  854.22   380.3  854.81
   389.6  854.85   398.9  854.61   408.4   854.1   427.4  852.36   436.9  851.71
   474.9   850.7   484.4  850.31   493.9  849.51   512.9  846.78   522.4  846.91
   531.9  850.07   541.4  856.56   550.9  863.77   560.4  869.83   569.9  874.69
   579.4  878.61   589.2  882.45   618.7  893.78   628.6  897.73   638.4   901.8
#Mann= 3 , 0 , 0
       0      .1       0   493.9    .045       0   531.9      .1       0
Bank Sta=493.9,531.9
XS Rating Curve= 0 ,0
Exp/Cntr=0.3,0.1

Type RM Length L Ch R = 1 ,96635.9 ,70.3,67.3,64.1
XS GIS Cut Line= 4
     1889812.006      496769.108     1889667.603      496877.765
     1889452.145      496881.489     1889373.812      496919.822
#Sta/Elev= 30
       0   890.6     9.5  887.64    57.1  873.16    66.6  870.13    76.1  866.97
    85.6  863.67    95.1  860.92   104.6   859.3   114.1  858.68   152.2  856.76
   180.7   855.2   219.9  853.28   268.9  851.08   288.5  850.44   298.3   849.1
   303.3847.8835     308  846.74   317.8  845.94   327.6  847.56   337.4  849.74
   347.2  850.94   366.8  851.64   376.6  853.21   386.4   856.2   396.2  859.64
   415.6  867.44   425.3  871.46   444.7  879.96   454.4  884.36   483.4  898.18
#Mann= 3 , 0 , 0
       0      .1       0   303.3    .045       0   327.6      .1       0
Bank Sta=303.3,327.6
XS Rating Curve= 0 ,0
Exp/Cntr=0.3,0.1

Type RM Length L Ch R = 1 ,96568.5 ,41.8,41.9,42.2
XS GIS Cut Line= 3
     1889784.922      496712.163     1889675.153       496794.48
     1889332.423      496844.406
#Sta/Elev= 30
       0  900.86     9.8  896.88    19.6  892.66    58.8  874.99    78.4  866.42
    88.2  862.49      98  859.55   107.8  858.01   117.6  857.36   137.2  856.54
   175.7   854.7   194.9  853.66   204.6  853.01   223.8  851.32   233.4  850.23
     243  848.78   252.6  846.97   262.3  845.48   271.9  845.11   281.5  846.04
   291.1  847.88   300.8  849.32   310.4  849.84   358.5  850.58   368.1  851.07
   377.7  852.67   387.4  855.71   435.4  874.67   445.1  878.56   483.6  894.62
#Mann= 3 , 0 , 0
       0      .1       0   252.6    .045       0   281.5      .1       0
Bank Sta=252.6,281.5
XS Rating Curve= 0 ,0
Exp/Cntr=0.3,0.1

Type RM Length L Ch R = 1 ,96526.6 ,271.9,266,259.8
XS GIS Cut Line= 3
     1889776.312      496660.517     1889649.125       496756.87
     1889325.201      496804.406
#Sta/Elev= 30
       0  911.81    18.8  904.54    28.2  900.16    46.9  889.12    56.3  884.08
    84.5     870    93.9  865.58   103.2  861.54   112.6  858.67     122  857.07
   131.4  856.32   159.6  854.88   169.2  854.25   188.4  852.69   207.7  850.78
     227  848.64   246.2  845.96   255.9  845.05   265.5  844.94   275.1  846.14
   284.7   847.9   294.4  848.88   332.9  849.97     381  850.83   390.7  851.21
   400.3  852.53   409.9  855.17   419.6  858.55   467.7  876.07     487  883.86
#Mann= 3 , 0 , 0
       0      .1       0   246.2    .045       0   275.1      .1       0
Bank Sta=246.2,275.1
XS Rating Curve= 0 ,0
Exp/Cntr=0.3,0.1

Type RM Length L Ch R = 1 ,96260.6 ,472.9,450.6,427.4
XS GIS Cut Line= 4
     1889662.166      496407.892     1889554.486       496485.74
     1889301.055      496597.336     1889216.749      496712.753
#Sta/Elev= 30
       0  945.51      19   938.2      38  930.56    47.4  926.26      57  919.72
    66.4  911.19    94.9  882.77   104.4  873.46   113.9   864.3   123.4  856.09
   132.9  850.85   142.4  849.43   161.5  848.28   171.1  847.44   187.9844.9722
   190.2  844.62   199.7  843.92   209.3  844.14   217.9 845.425   228.4  847.12
   237.9  847.99   247.5  848.38   352.5  851.18   400.2  852.28   419.3  852.46
   447.9  852.38   457.4  853.45     467  855.93   514.6  874.24   552.7  889.18
#Mann= 3 , 0 , 0
       0      .1       0   187.9    .045       0   217.9      .1       0
Bank Sta=187.9,217.9
XS Rating Curve= 0 ,0
Exp/Cntr=0.3,0.1

Type RM Length L Ch R = 1 ,95810   ,450.2,430.8,410.9
XS GIS Cut Line= 3
     1889190.636      496061.314     1889115.983      496506.626
     1889140.246      496690.543
#Sta/Elev= 30
       0   954.8    58.9  921.32    98.2  899.35     157  867.46   176.7   857.1
   186.5  852.32   196.3   848.8   206.1  846.69   231.4  842.27   235.6  841.58
   245.4   840.9   255.2  841.79   261.4843.4222   274.8  846.75   284.7  847.42
   304.3  847.42   353.4  846.63     373  846.77   412.3  847.77   451.5  850.42
   480.8  849.68   490.6  850.05   510.1  850.17   519.9  850.66   529.6  853.26
   549.2  861.85   568.7  869.87   578.4  872.64   607.8  878.77     637   885.7
#Mann= 3 , 0 , 0
       0      .1       0   231.4    .045       0   261.4      .1       0
Bank Sta=231.4,261.4
XS Rating Curve= 0 ,0
Exp/Cntr=0.3,0.1

Type RM Length L Ch R = 1 ,95379.2 ,374.9,378.2,381.3
XS GIS Cut Line= 3
     1888651.983      496264.154     1888879.413      496532.348
      1888983.58      496718.147
#Sta/Elev= 30
       0  933.08     9.8   925.1    19.5  916.54    29.3  909.16    39.1  902.84
    58.6  891.37    78.1     880   107.4  863.42     127  852.85   136.8  848.85
   163.2841.8032     166  841.07   175.8  839.42   185.6  840.12   193.2842.3073
   205.1  845.65   214.9  846.25   302.8  844.34   351.6  843.92   380.7  844.97
     400  845.16   448.5  847.94   458.2  848.94   467.8  850.54   506.6   857.9
   516.2  859.92   525.9  862.43   535.6  864.39     555  867.84   564.6  870.16
#Mann= 3 , 0 , 0
       0      .1       0   163.2    .045       0   193.2      .1       0
Bank Sta=163.2,193.2
XS Rating Curve= 0 ,0
Exp/Cntr=0.3,0.1

Type RM Length L Ch R = 1 ,95001   ,160.2,159.4,158.6
XS GIS Cut Line= 5
     1888478.465       496264.44     1888485.409       496474.51
     1888459.715      496610.447     1888514.576      496697.947
     1888526.381      496847.947
#Sta/Elev= 30
       0  889.59      86  882.47   143.3  876.13   191.1  869.88   200.6  868.16
   210.2  865.96   228.6  860.39   256.3  852.88   293.2  841.55   302.4  839.23
   311.6  838.64   348.5  840.39   367.3  840.59   376.7  839.05   383.6837.1121
   386.1  836.41   395.5  835.52   404.9  836.05   413.6838.2203   423.6  841.22
     433  842.19   508.2  840.55   517.6  840.68     527   842.4   545.8   848.8
   555.2  850.49   564.6  854.15   574.1  860.62   583.5  866.41   602.3  876.71
#Mann= 3 , 0 , 0
       0      .1       0   383.6    .045       0   413.6      .1       0
Bank Sta=383.6,413.6
XS Rating Curve= 0 ,0
Exp/Cntr=0.3,0.1

Type RM Length L Ch R = 1 ,94841.6 ,40.3,39.9,39.4
XS GIS Cut Line= 3
     1888131.242      496311.836     1888198.897      496509.102
     1888425.569      496847.263
#Sta/Elev= 30
       0  899.67      19  893.36    47.4  883.26    66.4  877.49    85.3  872.75
   151.7  858.13   161.2  855.59   180.1  849.86   189.6  847.68   227.9  843.58
     257  839.74   266.7  838.76   305.5   836.4   324.9  836.13   344.2  836.49
   441.2  841.45   450.9  841.28   467.1837.3892   470.2  836.54     480  835.08
   489.6  835.24   499.3  836.97   518.7  841.91   538.1  845.61   547.8  849.85
   557.5  855.08   567.2  858.24   576.9  860.37   586.6  862.97   615.6  873.99
#Mann= 3 , 0 , 0
       0      .1       0   467.1    .045       0   499.3      .1       0
Bank Sta=467.1,499.3
XS Rating Curve= 0 ,0
Exp/Cntr=0.3,0.1

Type RM Length L Ch R = 1 ,94801.8 ,196.1,210.8,225.2
XS GIS Cut Line= 2
     1888105.305      496437.821     1888392.235      496866.291
#Sta/Elev= 30
       0  873.71    29.2  865.07    48.6  859.12    77.8  850.83    87.6  848.25
    97.3  846.51   116.8  844.74   126.5  843.65   165.4  838.71   184.9   837.1
   194.6  836.52   204.3  836.17   223.8     836     253  836.66   330.8  840.62
   340.5  840.49   350.3   838.9   358.9836.9584   369.7  835.15   379.5  834.94
   389.2   835.8   398.9  838.03   408.6  841.64   418.4  846.33   437.8  856.69
   447.6  860.23   457.3  862.21     467  864.66   476.8  867.96   515.7  883.27
#Mann= 3 , 0 , 0
       0      .1       0   358.9    .045       0   389.2      .1       0
Bank Sta=358.9,389.2
XS Rating Curve= 0 ,0
Exp/Cntr=0.3,0.1

Type RM Length L Ch R = 1 ,94591   ,477.9,464.7,451.6
XS GIS Cut Line= 4
     1888039.749      496452.265     1888109.749      496566.154
     1888101.971      496827.821     1888156.416       496961.71
#Sta/Elev= 30
       0   883.2    19.1  875.82    28.6   872.3    66.8  858.55    85.9  851.59
    95.5  848.19     105  845.83   114.6  844.91   133.7  844.47   201.6   842.1
   240.3  840.91   259.7  840.38   269.4  840.22   298.5  840.09   308.2  839.57
   321.4836.7551   327.6   835.4   337.3  834.87     347     836   351.4837.2746
   356.7  838.81   366.4  842.93   385.8  852.93   395.5  856.47   405.1  859.26
   414.7  862.59   424.4  866.62   453.3  878.98   511.1  903.89     540  916.02
#Mann= 3 , 0 , 0
       0      .1       0   321.4    .045       0   351.4      .1       0
Bank Sta=321.4,351.4
XS Rating Curve= 0 ,0
Exp/Cntr=0.3,0.1

Type RM Length L Ch R = 1 ,94126.3 ,411.8,415.8,419.6
XS GIS Cut Line= 2
     1887553.466      496642.684     1887870.306      497158.309
#Sta/Elev= 30
       0  920.55    29.3  906.79      39  902.07    48.8  896.51    58.6     890
    87.8  870.07   117.1  850.36   126.9  843.61   136.7  836.66   146.4  831.84
   156.2  830.08   165.9  829.81   175.7  829.88   185.5  830.55   195.2  833.19
     205  835.12   214.8     836   283.1  837.55   390.4  840.47   400.2  840.98
     410  842.28   429.5  845.67   439.2  847.62     449  850.33   458.8   853.5
   527.1  876.73   546.6  883.59   566.2   890.7   585.7  898.27   605.2  906.52
#Mann= 3 , 0 , 0
       0      .1       0   146.4    .045       0   185.5      .1       0
Bank Sta=146.4,185.5
XS Rating Curve= 0 ,0
Exp/Cntr=0.3,0.1

Type RM Length L Ch R = 1 ,93710.5 ,265,262.1,258.9
XS GIS Cut Line= 4
     1887240.673      496872.232     1887274.936      496962.159
      1887340.19      497126.129     1887451.548      497344.884
#Sta/Elev= 27
       0  883.44     9.6  879.75    28.9  872.03    48.1  864.13    86.6  848.17
     106  840.26   115.8  836.11   125.6  831.66   135.4   828.5   145.2   827.3
   155.1  827.47   164.9  830.34   174.7  835.03   184.5  836.95   194.3  837.17
   243.3  837.07   292.4  836.82   351.3   836.8   380.7  836.99   390.5   837.3
   400.4  837.96   410.2  838.88   449.4  842.81   459.3  844.29   469.1   846.8
   488.7   852.9   518.2  862.44
#Mann= 3 , 0 , 0
       0      .1       0   135.4    .045       0   164.9      .1       0
Bank Sta=135.4,164.9
XS Rating Curve= 0 ,0
Exp/Cntr=0.3,0.1
